HEC-RAS study ROCKCK.prj: ROCKCK

--- ROCKCK.g01 (geometry) --- (continued)

Type RM Length L Ch R = 1 ,9866.2  ,224.9,225.7,226.2
XS GIS Cut Line= 2
     1732194.398      403007.377     1732197.002      403511.283
#Sta/Elev= 30
       0  760.12      12  752.74      36  741.01      56  729.51      64  722.45
      76     707      80  702.86      84  700.44     100  697.32     108  697.21
  115.17698.6521     128   703.4  144.71704.0218     156  703.48     160  702.46
     164  701.12     172  695.55   179.8  693.78     188  693.54   194.8  693.85
     200  694.52     216  702.88  233.31703.3233  262.85703.7639  292.38704.8719
   319.9  705.04   399.9  709.38   447.9  714.13   475.9  718.57   503.9  720.93
#Mann= 8 ,-1 , 0
       0     .12       0  115.17    .016       0  144.71     .12       0
   179.8    .045       0   194.8     .12       0  233.31     .06       0
  262.85     .12       0  292.38     .06       0
#XS Ineff= 2 , 0
          145.57   705.2
Permanent Ineff=
       F       F
Bank Sta=179.8,194.8
XS Rating Curve= 0 ,0
Exp/Cntr=0.3,0.1

Type RM Length L Ch R = 1 ,9640.6  ,294.7,297.9,300.9
XS GIS Cut Line= 2
     1731973.044      402985.242     1731966.533      403524.304
#Sta/Elev= 30
       0  785.58      16  775.15    35.9  760.66    63.9   745.5    71.9   740.1
    75.9   736.6    91.8  719.77    95.8  716.22   111.8  704.74   115.8  702.21
   119.8  701.45  124.49701.9669   131.8  702.34   151.8  701.98   167.7  701.35
   171.7   700.8   175.7  699.43   185.8   693.4   187.7  692.52   191.7  692.02
   195.7  692.12   200.8  692.93   203.7  693.78   215.6  699.96   219.6  701.16
   247.6  703.12   323.5  705.26   383.4   705.1   521.3707.5705   539.1  707.97
#Mann= 5 ,-1 , 0
       0     .12       0  124.49    .016       0   185.8    .045       0
   200.8    .016       0   521.3     .08       0
#XS Ineff= 2 , 0
          147.11  705.41
Permanent Ineff=
       F       F
Bank Sta=185.8,200.8
XS Rating Curve= 0 ,0
Exp/Cntr=0.3,0.1

Type RM Length L Ch R = 1 ,9342.7  ,150.3,153.6,156.8
XS GIS Cut Line= 3
     1731777.983      402892.099     1731692.046      403053.558
     1731649.077      403510.589
#Sta/Elev= 30
       0  815.01    31.8   798.3    51.7  785.77    67.6     778    99.4  755.96
   131.2  738.38   151.1  723.03     163  707.38     171  701.25   178.9  698.68
  192.87698.5172   206.8  700.08  222.54700.1606   270.7  699.53  311.54696.0696
   334.7  691.48   342.6  691.12   349.7  691.34   352.3691.7922   354.6  692.35
   362.5  698.57   366.5  699.92  459.86701.1673   482.3  700.55   538.2  702.89
  578.53703.2365   590.1  703.33     602  707.04     626  712.37     642  712.92
#Mann= 9 ,-1 , 0
       0     .12       0  192.87    .016       0  222.54     .08       0
  311.54     .12       0   334.7    .045       0   349.7     .12       0
   352.3     .08       0  459.86     .06       0  578.53     .12       0
#XS Ineff= 2 , 0
       0  222.54  703.75   381.9       0  703.75
Permanent Ineff=
       F       F
Bank Sta=334.7,349.7
XS Rating Curve= 0 ,0
Exp/Cntr=0.3,0.1

Type RM Length L Ch R = 1 ,9189.1  ,138.5,137.3,136.6
XS GIS Cut Line= 3
     1731593.238      402816.857     1731516.415      403238.732
      1731476.95      403486.544
#Sta/Elev= 30
       0  827.48    27.8  811.87    67.5  785.98    87.4  775.33   127.1   751.2
   170.7   730.8   190.6  715.41   202.5  700.69   206.5  697.22   210.4  696.13
   218.4  696.13  250.68698.9818  280.71698.8438   309.7   699.1  340.75698.2775
   345.4  698.28   349.4   696.6   357.3  691.15   359.2     691   373.2  690.49
   374.2  690.55   381.2   691.3   385.1  693.04   393.1  698.25  400.79 700.558
  610.25  704.06  640.16704.7393   643.9  705.16   651.9   709.1   679.8  718.71
#Mann= 9 ,-1 , 0
       0     .12       0  250.68    .016       0  280.71     .06       0
  340.75     .12       0   359.2    .045       0   374.2     .06       0
  400.79     .08       0  610.25     .06       0  640.16     .12       0
#XS Ineff= 2 , 0
       0     280     720               0
Permanent Ineff=
       F       F
Bank Sta=359.2,374.2
XS Rating Curve= 0 ,0
Exp/Cntr=0.3,0.1

Type RM Length L Ch R = 1 ,9051.8  ,115.1,128.4,141.2
XS GIS Cut Line= 2
     1731461.325      402773.002     1731348.044       403421.44
#Sta/Elev= 30
       0   851.5      20  836.42    27.9  828.95    51.9  810.24    79.8  795.24
   139.6  757.29   155.6  746.02   167.6  734.98   175.5  728.91   195.5  717.98
   211.4  702.55   219.4  696.76   223.4  695.05   231.4  694.22   264.9  697.15
   283.2  698.41  294.88697.5984  324.87 696.145   347.1  693.73   359.6  689.37
     367  688.55   374.6  689.28     387  694.57   398.9  697.38   444.8   699.4
  564.73701.8821   602.4  702.23  624.69704.1577   642.3  706.52   658.3   711.1
#Mann= 9 ,-1 , 0
       0     .12       0   264.9    .016       0  294.88     .06       0
  324.87     .12       0   359.6    .045       0   374.6     .12       0
   444.8     .06       0  564.73     .12       0  624.69     .06       0
#XS Ineff= 2 , 0
       0   287.2     720               0
Permanent Ineff=
       F       F
Bank Sta=359.6,374.6
XS Rating Curve= 0 ,0
Exp/Cntr=0.3,0.1

Type RM Length L Ch R = 1 ,8923.4  ,169,171.7,174.3
XS GIS Cut Line= 3
     1731381.898       402765.19     1731361.065      402935.762
     1731144.919      403331.596
#Sta/Elev= 30
       0  847.37      28  826.41      36   821.4    59.9  804.48    71.9  799.81
    75.9  797.42   111.9  772.69   127.9  762.53   143.9  750.21   163.8  730.42
   171.8   724.3   191.8   711.4   195.8  707.91   203.8  697.58   207.8  694.51
   215.7  692.97  250.06696.2827   267.6  697.53  283.72697.4625   291.6  696.08
   299.6  692.06   309.7  689.09   319.5  688.54   324.7  688.76   339.5  692.27
   359.4  693.73  384.67696.6857     535  701.37     563  700.67   622.8  706.36
#Mann= 6 ,-1 , 0
       0     .12       0  250.06    .016       0  283.72     .12       0
   309.7    .045       0   324.7     .12       0  384.67     .06       0
#XS Ineff= 2 , 0
       0   275.6     720               0
Permanent Ineff=
       F       F
Bank Sta=309.7,324.7
XS Rating Curve= 0 ,0
Exp/Cntr=0.3,0.1

Type RM Length L Ch R = 1 ,8751.7  ,326.1,332.7,339.2
XS GIS Cut Line= 2
     1731311.988      402713.992     1730998.186      403204.877
#Sta/Elev= 30
       0  867.09    39.9  843.88    47.9  836.54    63.8  824.74    95.8  803.28
   115.7  791.21   171.6  750.93   175.6  746.16   183.6  733.68   195.5   719.3
   203.5  708.39   211.5   700.6   219.5  696.21   227.5  693.96   231.4  693.28
  239.54694.1854  274.59696.4801   283.3   695.8   295.3  691.12     312  687.83
   319.2  687.77     327  688.63   335.2  691.36  379.75 697.557  420.54698.0054
     443  698.45  449.86699.7348   462.9  702.34  484.92703.0377   582.6  704.55
#Mann= 9 ,-1 , 0
       0     .12       0  239.54    .016       0  274.59     .06       0
     312    .045       0     327     .06       0  379.75    .016       0
  420.54     .06       0  449.86    .016       0  484.92     .06       0
#XS Ineff= 2 , 0
       0  270.18     740               0
Permanent Ineff=
       F       F
Bank Sta=312,327
XS Rating Curve= 0 ,0
Exp/Cntr=0.3,0.1

Type RM Length L Ch R = 1 ,8419    ,304.9,302.5,299.7
XS GIS Cut Line= 3
     1731172.263      402598.523     1730986.065      402662.325
     1730686.585      402987.846
#Sta/Elev= 30
       0  828.29    15.8  818.06    31.5  806.18    43.3  800.42    55.1  796.57
    70.9  788.82   118.1  756.01   137.8  744.54   149.6  736.54   177.1  716.74
   196.8  706.63   204.8  703.96   216.8  698.42   244.6  695.58   252.6  693.32
  260.35693.3813  300.48 693.228  311.73692.7452   328.3  691.93   342.2  686.42
   352.2  685.47   357.2  685.79   368.2  690.14  380.75697.1625   392.1  698.84
     428  701.05   499.7  700.31   603.3  701.91   623.2  703.04   639.2  707.05
#Mann= 7 ,-1 , 0
       0     .12       0  260.35    .016       0  300.48     .06       0
  311.73     .12       0   342.2    .045       0   357.2     .12       0
  380.75     .06       0
Bank Sta=342.2,357.2
XS Rating Curve= 0 ,0
Exp/Cntr=0.3,0.1

Type RM Length L Ch R = 1 ,8116.5  ,203.4,203.4,203.4
XS GIS Cut Line= 3
      1730892.92      402297.085     1730693.564       402545.48
     1730494.209      402793.874
#Sta/Elev= 30
       0  791.19    11.9  784.77    35.8  765.24    47.8  757.56    59.7  746.15
    79.6  731.98    91.6  721.53    99.5  717.33   111.5  712.63   139.3  695.58
   151.3  694.59   195.1  695.68  258.61691.8738   290.6  691.55   294.6  690.49
  301.04686.6384   305.8  684.57   318.5  684.12   320.8  684.14   326.5  684.67
   346.4   692.5   354.3  694.26   394.1  694.58  414.66697.6697   485.7  695.79
  528.27  695.76  566.14696.0726  588.91696.3235  604.01696.4811     637   697.1
#Mann= 10 ,-1 , 0
       0     .12       0  258.61    .016       0  301.04     .12       0
   305.8    .045       0   320.8     .12       0  414.66     .06       0
  528.27    .016       0  566.14     .06       0  588.91     .08       0
  604.01     .06       0
Bank Sta=305.8,320.8
XS Rating Curve= 0 ,0
Exp/Cntr=0.3,0.1

Type RM Length L Ch R = 1 ,7913.2  ,254.6,257.3,259.8
XS GIS Cut Line= 3
      1730743.18      402159.065     1730543.825      402407.459
      1730344.47      402655.853
#Sta/Elev= 30
       0   802.7       8  798.37    31.8  781.75    47.8  768.96    67.7  756.43
   103.5  725.77   119.4  717.47   143.3  701.78   155.3  695.54   159.2  692.03
   163.2  690.43   175.2  691.54     207  691.78  255.32690.2287   286.6   690.5
   294.6  689.58   302.5686.7067   313.4  683.51   330.4  683.34  335.06683.4968
   338.4  684.24   346.4  690.25   350.4  691.26  402.28692.3027   441.9  694.87
  515.89693.5971  553.76693.3909   605.2  694.12  629.51695.5902     637  695.75
#Mann= 9 ,-1 , 0
       0     .12       0  255.32    .016       0   302.5     .12       0
   313.4    .045       0  335.06     .12       0  402.28     .06       0
  515.89    .016       0  553.76     .06       0  629.51     .08       0
#XS Ineff= 2 , 0
       0     207     700               0
Permanent Ineff=
       F       F
Bank Sta=313.4,335.06
XS Rating Curve= 0 ,0
Exp/Cntr=0.3,0.1

Type RM Length L Ch R = 1 ,7655.9  ,325.2,324.4,322.6
XS GIS Cut Line= 2
     1730548.817      402024.912     1730050.119      402563.974
#Sta/Elev= 30
       0  803.42      20  792.12    43.9  775.61    75.8  755.85   111.8  732.16
   127.7  720.25   159.6  691.77   167.6  689.27  210.07687.4294   215.5  686.85
   231.5  689.03  253.57688.8527   263.4  687.34   271.4   683.7   277.3  682.39
   283.4  682.04   292.3  682.26   303.3  683.43   311.3  689.47   319.3  690.85
  427.53 690.846  449.21690.6492  489.45691.6091  529.69692.4333  558.01693.3303
   614.6     696   634.6  703.92   670.5  712.56  688.48719.1356   734.4  741.96
#Mann= 11 ,-1 , 0
       0     .12       0  210.07    .016       0  253.57     .12       0
   277.3    .045       0   292.3     .12       0  427.53     .06       0
  449.21    .016       0  489.45     .06       0  529.69     .08       0
  558.01     .06       0  688.48     .12       0
Bank Sta=277.3,292.3
XS Rating Curve= 0 ,0
Exp/Cntr=0.3,0.1

Type RM Length L Ch R = 1 ,7331.5  ,227.3,228.7,230
XS GIS Cut Line= 3
     1730468.238      401879.356     1730209.123      401913.211
     1729864.071      402318.159
#Sta/Elev= 30
       0  829.79   106.9  786.43   130.7  775.06   178.2  751.12   201.9  736.73
   261.3  703.39   285.1  692.12     305  687.62  336.85 687.055   352.6  687.74
  375.65685.8523   380.4  685.22     392  681.35   408.2  680.56   416.2  681.58
   424.1  684.54     432  685.59  503.99687.2027   519.4  688.55  549.53688.7633
  569.67689.2301   590.8  690.27  608.48689.9266   638.5  689.55   686.1  692.93
     706  697.57  724.89 705.805   737.8  713.17   753.6  720.75   793.3   748.7
#Mann= 10 ,-1 , 0
       0     .12       0  336.85    .016       0  375.65     .12       0
     392    .045       0   416.2     .06       0  503.99     .12       0
  549.53     .06       0  569.67     .12       0  608.48     .06       0
  724.89     .12       0
#XS Ineff= 2 , 0
                          518.61          692.24
Permanent Ineff=
       F       F
Bank Sta=392,416.2
XS Rating Curve= 0 ,0
Exp/Cntr=0.3,0.1

Type RM Length L Ch R = 1 ,7102.8  ,198.3,193.2,187.8
XS GIS Cut Line= 3
     1730153.134      401535.606     1730089.332      401715.294
     1729715.634      402124.148
#Sta/Elev= 30
       0   782.2    19.9  773.97    47.7   759.1   119.2  724.33   131.1  716.22
  148.29706.5009   158.9  699.56   162.9  697.83   170.8  696.41   298.3  691.04
   314.2  689.58   326.2  686.74  333.97686.7883  376.65683.6196   390.8  679.53
   397.9  679.05   405.8  679.31   425.8  683.93  496.69684.8895  576.72684.4056
     621  684.12  640.41685.3235     649  688.74   660.9  695.85   672.9  700.41
  684.19706.8375   700.8  714.46   716.7  724.31   728.6  730.01   744.6  741.81
#Mann= 10 ,-1 , 0
       0     .12       0  148.29     .06       0  333.97    .016       0
  376.65     .12       0   390.8    .045       0   405.8     .12       0
  496.69     .06       0  576.72     .12       0  640.41     .06       0
  684.19     .12       0
Bank Sta=390.8,405.8
XS Rating Curve= 0 ,0
Exp/Cntr=0.3,0.1

Type RM Length L Ch R = 1 ,6909.6  ,65.8,65.8,65.8
XS GIS Cut Line= 3
     1729995.061      401467.724     1729651.311      401966.423
     1729578.394      402008.089
#Sta/Elev= 30
       0  769.36    35.9  754.11    71.7  735.69    87.7   731.1    99.6     729
   115.6  722.52   123.5  717.84   147.4   698.6   163.4  689.31   187.3  686.05
  264.44 684.714   306.8  684.17  316.48  681.58     321  679.37   326.8  677.75
     336  678.62   354.6  683.29  368.52683.7356  431.54683.7943   466.2  684.87
   553.9  683.59   565.8   685.7   569.8  687.26   589.8     703   593.7  704.65
   601.7  704.84   605.7  706.26   637.7  721.47   653.7   735.4   689.7  759.64
#Mann= 7 ,-1 , 0
       0     .12       0  264.44    .016       0  316.48     .12       0
     321    .045       0     336     .12       0  368.52     .06       0
  431.54     .12       0
Bank Sta=321,336
XS Rating Curve= 0 ,0
Exp/Cntr=0.3,0.1

Type RM Length L Ch R = 1 ,6843.8  ,184,180.1,176.5
XS GIS Cut Line= 3
      1729936.12      401437.864      1729592.37      401936.562
     1729519.453      401978.228
#Sta/Elev= 30
       0  756.48    35.9  743.87    87.7   727.3    95.6  722.84   111.6   710.2
   119.5  705.44   127.5  699.01   131.5  696.64   143.4  693.55   151.4  689.42
   171.4  687.28  212.63685.3043  252.57684.3336     271  684.94  288.45684.1974
   302.8  683.25  316.71679.4537   316.8  679.42   322.8  678.18   331.8  678.77
   342.7  682.37   350.7  683.02   450.3   684.8  503.68683.4863     534  682.94
   541.9   684.2   549.9  692.01   557.9  697.75   593.7  713.76   689.7  770.85
#Mann= 8 ,-1 , 0
       0     .12       0  212.63     .06       0  252.57    .016       0
  288.45     .08       0  316.71     .06       0   316.8    .045       0
   331.8     .06       0  503.68     .12       0
Bank Sta=316.8,331.8
XS Rating Curve= 0 ,0
Exp/Cntr=0.3,0.1

Type RM Length L Ch R = 1 ,6663.7  ,158.9,152.2,143.8
XS GIS Cut Line= 3
     1729752.471      401333.158     1729480.336      401826.648
     1729425.648      401864.408
#Sta/Elev= 30
       0  760.88      48  742.95    71.9  735.25    83.9  730.01    95.9  722.81
   107.9  712.87   143.9  687.38   155.9  685.06  188.41682.6708  255.87681.3807
   275.8  683.37  297.73 682.779   303.8  682.05   313.1  678.58   319.8  678.22
   328.1   678.6   347.7   681.3   371.7   681.2   403.7  682.61   467.6  682.12
   483.6  685.44  491.97686.1579   515.6  689.42   523.6  691.62   527.6  693.47
   539.6  702.02  559.43714.2648  587.02733.2559   610.5  748.55     630  759.66
#Mann= 9 ,-1 , 0
       0     .12       0  188.41     .06       0  255.87    .016       0
  297.73     .12       0   313.1    .045       0   328.1     .06       0
  491.97     .12       0  559.43     .06       0  587.02     .12       0
Bank Sta=313.1,328.1
XS Rating Curve= 0 ,0
Exp/Cntr=0.3,0.1

Type RM Length L Ch R = 1 ,6511.5  ,144.2,143.5,142.9
XS GIS Cut Line= 2
     1729557.442      401235.774     1729366.825      401844.003
#Sta/Elev= 30
       0  799.64    31.9  791.11    59.8  780.98    75.7  769.02    91.6  759.41
   111.5  743.06   147.4  721.43   159.4  712.33   183.2  691.07   195.2  684.15
   203.2  681.85   223.1  680.78     255  679.87  274.96680.8195  305.91682.7856
   330.6  682.13  336.86680.3279   340.4  678.94   342.6  678.36   355.4  678.53
   394.4  682.99  460.67 682.865   474.1  684.13     498  689.56   521.9  697.04
   541.8  708.05   557.7   718.3   577.6  728.12   593.6  738.92   637.4  764.26
#Mann= 7 ,-1 , 0
       0     .12       0  274.96     .08       0  305.91    .016       0
  336.86     .06       0   340.4    .045       0   355.4     .06       0
  460.67     .12       0
Bank Sta=340.4,355.4
XS Rating Curve= 0 ,0
Exp/Cntr=0.3,0.1

Type RM Length L Ch R = 1 ,6368    ,40.5,40.4,40.5
XS GIS Cut Line= 2
     1729400.813      401239.322     1729235.449      401799.218
#Sta/Elev= 30
       0  773.14      12  768.91      28  761.26      56  746.07      84  729.64
     128  699.47     144  692.23   167.9  686.24   179.9  684.66   211.9  682.22
   223.9  680.03  239.09 680.841  269.88681.5857   279.9  680.75   291.4  677.34
   299.9  677.23   306.4  677.57   308.8677.8445   319.9  682.13  331.48683.9143
  413.07689.2853  423.86689.2798   471.8  694.62   503.8  696.31   507.8  698.06
  516.26707.0902   519.8  710.17   531.8  716.72   559.8   738.2   583.8  748.22
#Mann= 10 ,-1 , 0
       0     .12       0  239.09    .016       0  269.88     .06       0
   291.4    .045       0   306.4     .06       0   308.8    .016       0
  331.48     .06       0  413.07    .016       0  423.86     .06       0
  516.26     .12       0
Bank Sta=291.4,306.4
XS Rating Curve= 0 ,0
Exp/Cntr=0.3,0.1

Type RM Length L Ch R = 1 ,6327.5  ,81.2,76.9,72.3
XS GIS Cut Line= 2
     1729362.619      401226.301     1729197.254      401786.197
#Sta/Elev= 30
       0   771.1      32  756.68      48  748.37      72   733.6     120  708.63
     140  694.66     156  687.91   175.9  684.76   211.9  682.24   223.9  679.75
  252.67681.2281   279.9  681.38  283.46680.0539   289.8  677.51   299.9  676.71
   304.8  677.01  314.26679.4741   319.9  682.73   323.9  683.81   382.5 687.078
  406.65688.5662   463.8  691.43  486.77695.2915  499.04695.4167   507.8  696.25
   515.8   699.4   531.8  712.54   543.8   719.7   555.8  731.38   583.8  744.17
#Mann= 10 ,-1 , 0
       0     .12       0  252.67    .016       0  283.46     .06       0
   289.8    .045       0   304.8     .06       0  314.26    .016       0
   382.5     .06       0  406.65    .016       0  486.77     .08       0
  499.04     .12       0
Bank Sta=289.8,304.8
XS Rating Curve= 0 ,0
Exp/Cntr=0.3,0.1

Type RM Length L Ch R = 1 ,6250.6  ,76.7,76.7,76.7
XS GIS Cut Line= 2
     1729259.554      401175.364      1729152.56      401803.719
#Sta/Elev= 30
       0  785.99    19.9  774.85    55.8  757.13    99.6  737.56   111.5  730.73
   131.5  716.01   155.4  703.54   175.3  689.97   183.2   686.1   195.2  683.15
   227.1  681.68     243  679.01  267.52680.6866  297.48 680.448   304.3  677.88
   310.7  676.44   322.7  677.23   334.6  681.83   357.4684.7954  447.28690.6559
   507.2692.9888   529.8  695.55  537.16697.5632   545.8  699.53   549.8   701.5
   561.7  712.09   581.6  723.34   593.6  731.78   613.5  739.48   637.4  745.76
#Mann= 9 ,-1 , 0
       0     .12       0  267.52    .016       0  297.48     .12       0
   304.3    .045       0   322.7     .12       0   357.4     .06       0
  447.28     .08       0   507.2     .06       0  537.16     .12       0
Bank Sta=304.3,322.7
XS Rating Curve= 0 ,0
Exp/Cntr=0.3,0.1

Type RM Length L Ch R = 1 ,6173.9  ,55.8,55.8,55.8
XS GIS Cut Line= 2
     1729183.165      401169.287     1729076.171      401797.642
#Sta/Elev= 30
       0  774.77    23.9  760.32    51.8   748.8    71.7  737.78    91.6  728.54
   107.6  724.18   131.5  720.32   139.4  717.69   151.4  710.95   175.3  690.79
   183.2  686.54   191.2  684.24   215.1  682.57     235  679.08  243.72 679.684
   286.8  680.42   299.3  676.28   306.8  675.89   314.3  676.85   322.7  679.59
  363.56681.7921   402.4  684.06   422.3  687.94  456.13691.0437   483.4694.4695
   525.8  698.75  543.32704.5086   565.7  710.16   601.6  717.57   637.4  723.12
#Mann= 8 ,-1 , 0
       0     .12       0  243.72    .016       0   299.3    .045       0
   314.3    .016       0  363.56     .06       0  456.13    .016       0
   483.4     .06       0  543.32     .12       0
Bank Sta=299.3,314.3
XS Rating Curve= 0 ,0
Exp/Cntr=0.3,0.1

Type RM Length L Ch R = 1 ,6118.1  ,84,84,84
XS GIS Cut Line= 2
     1729129.346      401155.399     1729022.352      401783.754
#Sta/Elev= 30
       0  781.29    15.9  768.61    39.8   752.9    63.7  738.96    79.7  731.02
    91.6  726.79   115.5  720.76   143.4  716.23   147.4   714.8   163.3  707.04
   187.2   697.3   203.2  685.55   215.1  680.69     235   678.9  257.81680.3781
  287.77 680.393   297.4   677.7   306.8   676.6   312.4  676.91  317.73677.9029
   330.6  681.16   390.4  682.64   410.3  685.48  467.53696.3223  487.41  698.15
   505.9  699.86   541.8  699.53  557.41702.9891   585.6  709.28   637.4  718.59
#Mann= 9 ,-1 , 0
       0     .12       0  257.81    .016       0  287.77     .12       0
   297.4    .045       0   312.4     .12       0  317.73     .06       0
  467.53    .016       0  487.41     .06       0  557.41     .12       0
Bank Sta=297.4,312.4
XS Rating Curve= 0 ,0
Exp/Cntr=0.3,0.1

Type RM Length L Ch R = 1 ,6034.1  ,214.8,214.2,213.3
XS GIS Cut Line= 2
     1729045.144      401152.794      1728938.15      401781.149
#Sta/Elev= 30
       0  771.63    27.9  751.19    43.8  741.02    59.8  731.94    79.7  722.58
   107.6   714.8   131.5  711.81   163.3  709.77   167.3  707.45   195.2  685.53
   203.2   680.5   211.1   678.8  230.49679.6888  260.45680.0222   270.9  679.91
   278.9  677.15   286.8  675.78   298.8  677.16   306.8   680.2  320.37680.8176
  410.26682.7378  440.22685.4822     498     694   513.9  697.58   530.1703.3545
   545.8  709.23   557.7  716.45   589.6  732.69   605.5     743   637.4  756.31
#Mann= 9 ,-1 , 0
       0     .12       0  230.49    .016       0  260.45     .12       0
   278.9    .045       0   298.8     .12       0  320.37     .06       0
  410.26     .12       0  440.22     .06       0   530.1     .12       0
#XS Ineff= 2 , 0
                          399.87          691.99
Permanent Ineff=
       F       F
Bank Sta=278.9,298.8
XS Rating Curve= 0 ,0
Exp/Cntr=0.3,0.1

Type RM Length L Ch R = 1 ,5819.9  ,299.1,300.9,302.1
XS GIS Cut Line= 3
     1728843.238      401099.408     1728749.488        401656.7
     1728780.738      401742.638
#Sta/Elev= 30
       0  766.93    11.9  761.14    35.8  746.03    47.8  742.54    67.7  740.31
    75.6  737.87    83.6   733.7    99.5  723.04   111.4   718.3   131.3  712.43
   155.2   707.1   167.2  700.64   183.1  695.06     203  692.18   218.9  682.72
  224.65681.2604   234.8  682.25  254.61 681.585   270.6  680.21  284.56675.9186
   286.5  675.55   294.5  674.95   302.5  675.34   326.3  684.34   338.3  686.72
   517.4  691.86   573.1  695.24     585  698.42   608.9  708.58   656.6  732.35
#Mann= 6 ,-1 , 0
       0     .12       0  224.65    .016       0  254.61     .12       0
  284.56     .06       0   286.5    .045       0   302.5     .06       0
Bank Sta=286.5,302.5
XS Rating Curve= 0 ,0
Exp/Cntr=0.3,0.1

Type RM Length L Ch R = 1 ,5518.9  ,225.9,219.8,213.3
XS GIS Cut Line= 3
     1728552.751      401069.069     1728495.521      401382.385
     1728438.249      401695.693
#Sta/Elev= 30
       0  823.87    19.9  809.76    55.7  790.77    71.7  783.76   107.5  763.32
   119.4  754.02   147.3  736.86   151.3   733.4   155.3  726.71  165.98704.5118
   167.2  702.02   171.2  696.51   175.2  695.06   183.1  695.54  205.15 694.861
     219  693.77     223  692.54   246.8  677.45   250.8  676.46   259.5  676.06
   274.5  675.62   278.7  676.29  286.08 679.346   302.6  685.27   310.5  686.88
   501.6   691.8   545.4  693.56   556.3695.0107   581.3  701.41     637   718.3
#Mann= 7 ,-1 , 0
       0     .12       0  165.98    .016       0  205.15     .12       0
   259.5    .045       0   278.7     .12       0  286.08     .06       0
   556.3     .12       0
Bank Sta=259.5,278.7
XS Rating Curve= 0 ,0
Exp/Cntr=0.3,0.1

Type RM Length L Ch R = 1 ,5299.1  ,106.9,105.3,104.8
XS GIS Cut Line= 3
     1728345.035      401016.839     1728289.479       401167.88
      1728282.04      401734.825
#Sta/Elev= 30
       0  838.11    31.4  814.96    39.2  810.88   149.2  739.14   153.1   735.9
     157  729.02   160.9  716.24   164.9  705.51  166.34704.3616   168.9  702.32
  195.88702.8633   208.8  700.32   244.8  684.81   268.7  681.96   283.9  674.55
   292.7  673.32   298.9  674.23  314.03 679.106   332.6  682.78   552.2  688.52
   568.2  690.39  579.87693.9543   588.2  696.74   600.2   698.6   612.1  707.14
   616.1  708.86  638.94 714.617     684  725.28     716  735.58   727.9  740.63
#Mann= 8 ,-1 , 0
       0     .12       0  166.34    .016       0  195.88     .12       0
   283.9    .045       0   298.9     .12       0  314.03     .06       0
  579.87    .016       0  638.94     .12       0
Bank Sta=283.9,298.9
XS Rating Curve= 0 ,0
Exp/Cntr=0.3,0.1

Type RM Length L Ch R = 1 ,5193.8  ,159.7,169,177
XS GIS Cut Line= 3
      1728275.53      400992.638     1728185.686      401186.648
     1728181.779      401736.127
#Sta/Elev= 30
       0  837.94    55.4   795.6      99  774.53   154.4  738.92   162.3  729.65
  166.53719.4144   170.2  709.75   174.2  702.81  199.08703.7335  201.16703.6055
   221.8  696.23   245.7  694.95  259.51689.3265   285.5  675.38   293.4  674.09
   301.4  673.73   313.5  674.14  318.58 675.508  377.66679.8616   508.5     687
  643.48687.3359   667.7  687.23   671.7  689.46   683.7  704.64   695.6  715.57
   711.5  724.53   723.5  727.24  732.09735.7673   747.4  750.37   763.3  760.28
#Mann= 11 ,-1 , 0
       0     .12       0  166.53    .016       0  199.08     .12       0
  201.16    .016       0  259.51     .12       0   293.4    .045       0
   313.5     .12       0  318.58     .06       0  377.66     .08       0
  643.48     .06       0  732.09     .12       0
#XS Ineff= 2 , 0
                           369.7          685.94
Permanent Ineff=
       F       F
Bank Sta=293.4,313.5
XS Rating Curve= 0 ,0
Exp/Cntr=0.3,0.1

Type RM Length L Ch R = 1 ,5024.8  ,225,223.2,221.4
XS GIS Cut Line= 3
     1728193.348      400958.506     1728050.119      401125.173
      1727919.91      401715.016
#Sta/Elev= 30
       0  840.75      16  828.75    63.9  799.52   183.8  733.11   187.8  728.82
   199.8  704.93  205.31703.4443   227.7  703.98  238.78702.0963   259.5  697.48
   287.3  686.68   299.2  676.66   304.4  674.09   315.1   673.3     327  673.69
  329.52674.4712  450.51683.0309  480.75683.9175     511684.5654  525.29684.9271
  601.74  686.58   662.3687.7966   700.6  688.18   704.6   689.6   716.5  700.03
  722.72708.1783   732.4  719.05   744.3  722.66   756.2  735.38   823.8  781.83
#Mann= 13 ,-1 , 0
       0     .12       0  205.31    .016       0  238.78     .12       0
   304.4    .045       0     327     .12       0  329.52     .06       0
  450.51     .08       0  480.75     .06       0     511     .08       0
  525.29     .06       0  601.74     .08       0   662.3     .06       0
  722.72     .12       0
Bank Sta=304.4,327
XS Rating Curve= 0 ,0
Exp/Cntr=0.3,0.1

Type RM Length L Ch R = 1 ,4801.6  ,348.7,329,308.1
XS GIS Cut Line= 2
     1727867.604      400862.325     1727718.298      401702.603
#Sta/Elev= 30
       0  799.16    75.8   767.5   159.5   721.3  177.36 706.776   187.4  700.75
  225.84699.9612   239.3  696.96   255.2  689.18   267.2  680.46   291.4  672.24
   295.1  672.08   311.1  672.35     323  675.95  345.83675.1451   430.7  679.66
   450.6  677.23   510.5  677.27   538.4  679.15   554.3  684.69  615.82685.3581
  675.81687.1833   693.9   686.8  705.81 693.717   713.9  698.18   725.8  714.93
   741.8  720.34   757.7  737.39   785.6  755.83   805.6  766.59   853.4  804.13
#Mann= 9 ,-1 , 0
       0     .12       0  177.36    .016       0  225.84     .12       0
   291.4    .045       0   311.1     .12       0  345.83     .06       0
  615.82     .08       0  675.81     .06       0  705.81     .12       0
Bank Sta=291.4,311.1
XS Rating Curve= 0 ,0
Exp/Cntr=0.3,0.1

Type RM Length L Ch R = 1 ,4472.6  ,319.3,295.8,278.3
XS GIS Cut Line= 4
     1727563.785      400832.811     1727426.632      400964.756
     1727683.576      401574.131      1727650.59      401711.283
#Sta/Elev= 30
       0  745.49    35.7  728.76    51.5  717.99    63.4  704.78    71.4   699.1
   107.7697.7703  113.28698.1937   150.3 704.054  192.26705.2997  256.37700.3992
  288.42698.0576   301.9  696.04  333.22682.2206   377.6  672.43   397.5  672.02
   401.5  672.42   413.4  675.55   453.2   673.2   469.2  676.14  485.26675.6952
  544.85678.0607   692.3  676.64   712.2   677.9   732.1   685.3     768  686.92
   811.8  684.65   823.8  692.07  833.33704.4611   922.2   767.4   992.7   820.6
#Mann= 13 ,-1 , 0
       0     .12       0   107.7     .08       0  113.28     .06       0
   150.3    .016       0  192.26     .08       0  256.37    .016       0
  288.42     .12       0  333.22    .016       0   377.6    .045       0
   401.5     .06       0  485.26     .08       0  544.85     .06       0
  833.33     .12       0
Bank Sta=377.6,401.5
XS Rating Curve= 0 ,0
Exp/Cntr=0.3,0.1

Type RM Length L Ch R = 1 ,4176.8  ,238.4,235.1,224.6
XS GIS Cut Line= 6
     1726982.187       401190.45      1727275.59      401298.089
     1727388.438      401403.992     1727428.368      401421.353
      1727579.41      401584.547     1727604.957      401727.013
#Sta/Elev= 30
       0  735.96    47.5   704.3   60.65702.7648    79.1  698.34   92.11701.1146
  123.57703.8348  155.03703.3277  186.49703.9282  217.95 703.031  280.88698.2812
  293.22697.2549  312.33695.2631  345.97691.9473  352.78691.2762   459.4  679.54
   475.2  676.59   484.8  670.26   487.1  669.48   499.8  669.59   530.7  674.08
  590.02673.5349  615.51673.4655   653.8  674.75   677.6  681.41   705.4  683.38
   709.4  686.91   721.3  719.68   737.1   734.6   838.8  806.58   877.9  827.32
#Mann= 16 ,-1 , 0
       0     .12       0   60.65     .06       0   92.11     .08       0
  123.57    .016       0  155.03     .08       0  186.49    .016       0
  217.95     .06       0  280.88     .12       0  293.22     .06       0
  312.33     .12       0  345.97     .06       0  352.78     .12       0
   484.8    .045       0   499.8     .12       0  590.02     .06       0
  615.51     .12       0
Bank Sta=484.8,499.8
XS Rating Curve= 0 ,0
Exp/Cntr=0.3,0.1

Type RM Length L Ch R = 1 ,3941.8  ,217.3,221.3,223.6
XS GIS Cut Line= 2
     1726921.424      401400.519     1727511.701      401716.492
#Sta/Elev= 30
       0  742.61      12  736.21    35.9  716.43    51.8  707.34   66.51 696.703
    71.7  693.89    79.7  692.46    91.7  692.89  100.01695.3917   111.6   697.7
  133.51 698.385   147.5  698.49   167.4  696.68  206.96699.1904   231.2  699.04
  267.51696.2814  301.02692.7598  368.02685.3854   426.4  678.58   476.2   669.5
   486.2  668.99   498.2  669.61   514.1   672.6   522.1  676.18     538  689.19
     554  707.34   561.9  714.64   617.7  751.94   633.7  760.95   669.5  783.34
#Mann= 10 ,-1 , 0
       0     .12       0   66.51     .06       0  100.01     .08       0
  133.51    .016       0  206.96     .06       0  267.51     .12       0
  301.02     .06       0  368.02     .12       0   476.2    .045       0
   498.2     .12       0
Bank Sta=476.2,498.2
XS Rating Curve= 0 ,0
Exp/Cntr=0.3,0.1

Type RM Length L Ch R = 1 ,3720.5  ,91.7,91.9,92
XS GIS Cut Line= 3
      1726806.84      401530.728      1727298.16      401831.075
     1727496.076      401839.755
#Sta/Elev= 30
       0  778.82      20  762.49      60  746.86      96  726.53     112  712.43
     136  695.36     152  689.43  164.13691.1031  168.41691.8822     180   694.1
  220.76696.1754  237.64694.1917  277.38697.7118  306.88697.3951   327.9  694.78
   371.9  674.95   387.9  670.03   395.9  669.25   407.9  671.05     427  668.88
   431.9  668.55   447.9  668.95   483.9  675.34   559.8   715.2   583.8  718.81
   599.6  718.32   607.6  720.52   655.1  744.17   674.9  750.33     774   810.7
#Mann= 9 ,-1 , 0
       0     .12       0  164.13     .06       0  168.41    .016       0
  220.76     .06       0  237.64    .016       0  277.38     .06       0
  306.88     .12       0     427    .045       0   447.9     .12       0
Bank Sta=427,447.9
XS Rating Curve= 0 ,0
Exp/Cntr=0.3,0.1

Type RM Length L Ch R = 1 ,3628.6  ,114.2,115.2,117.2
XS GIS Cut Line= 3
     1726723.446      401579.877     1727287.248       401931.44
      1727351.05       402049.93
#Sta/Elev= 30
       0  808.31    67.6  768.47   127.3  736.97  163.19707.9443   175.1  701.41
     191  689.19   210.9  688.29  232.81692.3538  236.36693.0764   274.5   695.9
  292.18693.3509  302.42694.2432  337.23697.6472   358.1  696.42   409.8   671.6
   421.7  669.24   445.6  669.67   449.6  668.98     468  669.88   481.4   671.1
   497.3  678.92   517.2  684.32   545.1  696.24     553  702.78   576.9  716.39
   636.6  720.97   648.5  718.69     708  749.22   763.4  762.18     799  784.11
#Mann= 9 ,-1 , 0
       0     .12       0  163.19     .06       0  232.81     .08       0
  236.36    .016       0  292.18     .06       0  302.42    .016       0
  337.23     .12       0   445.6    .045       0     468     .12       0
Bank Sta=445.6,468
XS Rating Curve= 0 ,0
Exp/Cntr=0.3,0.1

Type RM Length L Ch R = 1 ,3513.4  ,586.6,603.8,620.2
XS GIS Cut Line= 3
     1726688.195      401698.961     1726979.861      401864.326
     1727288.368      402092.538
#Sta/Elev= 30
       0  770.35      16  764.98    43.9  758.58    71.8  743.86   107.8  729.59
   123.7  716.88   135.7  710.94  165.76 689.078   183.6  687.07  199.71689.9139
  233.66694.6482   255.4  695.63   275.4   693.5  311.54697.3144   327.3  697.59
  335.54695.4326   375.3  683.25   387.2  673.87   395.2  669.82   407.2  668.16
   419.2  669.39   435.2  679.53   463.2  692.33  519.23699.3229   527.2  700.06
   543.1  709.07   563.9 712.546   579.1  721.09   655.1  755.05     719  793.77
#Mann= 10 ,-1 , 0
       0     .12       0  165.76     .06       0  199.71     .08       0
  233.66    .016       0  311.54     .06       0  335.54     .12       0
   395.2    .045       0   419.2     .12       0  519.23    .016       0
   563.9     .12       0
Bank Sta=395.2,419.2
XS Rating Curve= 0 ,0
Exp/Cntr=0.3,0.1

Type RM Length L Ch R = 1 ,2909.6  ,224.2,241.8,259.1
XS GIS Cut Line= 4
     1726396.623       401837.69     1726439.592      402075.971
     1726521.623      402215.294     1726843.238      402417.117
#Sta/Elev= 30
       0  843.65    87.3  789.91     123     764   142.9  751.97   158.8  735.18
   166.7  718.18   174.6  707.28  195.24696.8737  225.25695.3112   281.6  669.47
     307  664.77     321   664.7   324.9  664.79   340.7  670.55  375.99691.5364
  394.23702.3505   423.8  704.27  443.84701.8407  456.88703.5412  499.41704.6973
  526.62703.8591  561.49704.4297   579.7  702.92   595.6  698.13  610.54701.9163
   619.6  704.28   639.6  704.52   666.1  729.06   695.6  750.95   783.5  800.11
#Mann= 14 ,-1 , 0
       0     .12       0  195.24    .016       0  225.25     .12       0
     307    .045       0   324.9     .12       0  375.99     .08       0
  394.23    .016       0  443.84     .08       0  456.88    .016       0
  499.41     .06       0  526.62    .016       0  561.49     .12       0
  610.54    .016       0   666.1     .12       0
Bank Sta=307,324.9
XS Rating Curve= 0 ,0
Exp/Cntr=0.3,0.1

Type RM Length L Ch R = 1 ,2667.8  ,221.8,219.5,216.8
XS GIS Cut Line= 3
     1726220.692      401876.475     1726268.869      402384.287
     1726490.223      402536.631
#Sta/Elev= 30
       0  839.63    15.9  831.17    67.8  795.26    99.6  769.84   123.5  754.39
   135.5  749.32   159.4   735.6   163.4  732.16   175.3  715.52  183.72715.1647
   195.3  713.77   203.2  708.18  213.39698.4094   243.1  672.36   271.2   664.6
     275  664.45   286.2  664.66   302.9  671.36   330.8  669.16   434.4  669.15
   494.2  675.73   510.1  679.96  548.82 698.514  562.14704.8394   573.3  710.18
  584.67711.1642  656.38710.1226  666.33710.4099  770.52710.5739   778.8  710.37
#Mann= 11 ,-1 , 0
       0     .12       0  183.72    .016       0  213.39     .12       0
   271.2    .045       0   286.2     .12       0  548.82     .06       0
  562.14     .08       0  584.67    .016       0  656.38     .08       0
  666.33    .016       0  770.52     .06       0
#XS Ineff= 2 , 0
                          402.57          702.81
Permanent Ineff=
       F       F
Bank Sta=271.2,286.2
XS Rating Curve= 0 ,0
Exp/Cntr=0.3,0.1

Type RM Length L Ch R = 1 ,2448.3  ,190.4,189.1,185.1
XS GIS Cut Line= 2
     1725998.993      401954.454     1726090.828      402552.402
#Sta/Elev= 30
       0  817.68    47.8  785.24    75.6  764.66    91.5  754.14  106.15 746.482
   111.4  743.02   119.4  736.13   123.4  734.49  136.03734.6873   143.3  733.95
   147.3  732.05   175.1  708.72   187.1  697.47     203  676.44   210.9  668.36
   214.9   666.2   232.2  663.74   238.8   663.4   247.2  663.62   262.7  665.17
   274.6  672.08   278.6  673.19  285.44673.2316   318.4  673.73   330.3  674.66
   338.3  676.31   354.2  675.32   509.4  677.09   553.2  676.64     605  677.86
#Mann= 6 ,-1 , 0
       0     .12       0  106.15    .016       0  136.03     .12       0
   232.2    .045       0   247.2     .12       0  285.44     .08       0
Bank Sta=232.2,247.2
XS Rating Curve= 0 ,0
Exp/Cntr=0.3,0.1

Type RM Length L Ch R = 1 ,2259.2  ,182.8,182.9,183.4
XS GIS Cut Line= 3
      1725891.91       402002.95     1725843.299      402150.519
     1725930.104      402539.408
#Sta/Elev= 30
       0  767.19   28.31753.0993    35.8  749.41    43.8  743.76    47.8  742.44
    63.7  742.71    67.7  741.64    79.7  733.23   90.51727.4769   107.6  719.71
   119.5   712.5   159.4  691.52   167.3  685.79   179.3  674.95   183.3  672.44
   191.2  670.16   219.1  668.43   248.7   664.2     259  663.31   263.7  663.89
   290.8  668.92   298.8  672.49  304.08 673.292   322.7  672.71  364.61 674.135
  394.87674.8817  425.13676.9308   494.1   679.6  546.18678.6586   553.8  678.93
#Mann= 10 ,-1 , 0
       0     .12       0   28.31    .016       0   90.51     .12       0
   248.7    .045       0   263.7     .12       0  304.08     .06       0
  364.61     .08       0  394.87     .06       0  425.13     .08       0
  546.18    .016       0
#XS Ineff= 2 , 0
       0                   302.8       0  673.34
Permanent Ineff=
       F       F
Bank Sta=248.7,263.7
XS Rating Curve= 0 ,0
Exp/Cntr=0.3,0.1

Type RM Length L Ch R = 1 ,2076.3  ,124.3,129.2,134.1
XS GIS Cut Line= 3
     1725563.785       402065.45     1725659.271      402129.686
     1725759.965      402542.881
#Sta/Elev= 30
       0  727.42    67.5  721.99    83.3  718.55   115.1  704.05     127   697.5
     135  690.91   150.8  673.22   154.8  670.41   158.8  669.22   190.6  668.59
   226.4  669.37   250.2  668.56     282  669.24     286  668.69   293.9   665.4
     315  663.41   329.7  662.84   333.7  663.18   341.6  665.67   353.6  673.35
   365.5  675.43  377.11675.4066   401.3  674.66   425.1  674.84  468.31677.1996
   484.7  677.32   500.6  679.95   508.6  680.49   520.5  679.93   540.4  677.31
#Mann= 5 ,-1 , 0
       0     .12       0     315    .045       0   333.7     .12       0
  377.11     .08       0  468.31    .016       0
Bank Sta=315,333.7
XS Rating Curve= 0 ,0
Exp/Cntr=0.3,0.1

Type RM Length L Ch R = 1 ,1947.1  ,615.8,621.7,237.2
XS GIS Cut Line= 2
     1725568.298      402092.909     1725618.212      402564.915
#Sta/Elev= 30
       0  725.26      16  723.13    23.9  720.99    51.8  704.92    63.8  698.99
    67.8  696.08    75.8  688.14    87.8  673.82    91.7  670.03    95.7  667.89
   107.7  664.45   123.6  662.97   147.6  665.82   183.5  665.62   199.4  667.81
   235.3  667.77   255.3  668.55   279.2  668.19   283.2  667.35   287.5  664.17
   291.2  662.76   302.5  663.82   315.1  665.06   323.1  669.45   327.1  670.74
     335  671.47     347  673.87  382.08674.8026   406.8  674.83   474.6  677.02
#Mann= 4 ,-1 , 0
       0     .12       0   287.5    .045       0   302.5     .12       0
  382.08     .08       0
Bank Sta=287.5,302.5
XS Rating Curve= 0 ,0
Exp/Cntr=0.3,0.1

Type RM Length L Ch R = 1 ,1325.4  ,352.6,352.3,427.2
XS GIS Cut Line= 3
     1725458.706      402053.847     1725378.411      402124.377
     1725393.602       402491.13
#Sta/Elev= 30
       0  724.92     7.9  721.15    55.4  703.14      91  693.82   126.8  687.27
   138.8   681.9   150.8  672.55   154.8  670.49   166.7  665.87   174.7  663.43
   182.7  661.86   190.4  661.65   202.6  661.13   214.6  662.01   222.6  664.51
   238.5  666.25   242.5  666.18   250.5  663.71   254.5  663.36   266.5  667.21
   282.4  667.68   294.4   666.5   314.4  671.14   318.3  671.45   338.3  672.61
   358.2  672.83  396.55674.4561  426.11674.4199  455.67 675.291   473.9  676.02
#Mann= 6 ,-1 , 0
       0     .12       0   190.4    .045       0   214.6     .12       0
  396.55     .06       0  426.11     .08       0  455.67     .06       0
Bank Sta=190.4,214.6
XS Rating Curve= 0 ,0
Exp/Cntr=0.3,0.1

Type RM Length L Ch R = 1 ,973.1   ,231.4,213.1,180.5
XS GIS Cut Line= 3
     1725167.306      401955.902     1725091.785      402140.797
     1725154.285      402582.204
#Sta/Elev= 30
       0  725.12      40  723.39    83.9  719.47    95.9   717.4   119.8   710.2
  143.69704.3249   187.7  691.38   207.7  684.54   211.7   681.4   227.6  664.77
   231.6   661.2   235.6   659.6   239.5  659.59   250.7  660.17   255.4  660.66
   267.4  665.23   271.4  666.12   311.2  667.91   331.1  671.17     351  671.93
   366.9  674.32   370.9  674.23   378.8  672.55  385.97672.4037   398.8   672.3
   474.4  675.61   530.1  676.88   581.8  679.37   601.8   682.1   645.5  682.33
#Mann= 5 ,-1 , 0
       0     .06       0  143.69     .12       0   231.6    .045       0
   250.7     .12       0  385.97     .06       0
Bank Sta=231.6,250.7
XS Rating Curve= 0 ,0
Exp/Cntr=0.3,0.1

Type RM Length L Ch R = 1 ,760     ,113.8,113.7,122.5
XS GIS Cut Line= 4
     1724591.736      401887.831     1724714.349      402000.679
     1724995.382      402306.668     1725098.296      402596.527
#Sta/Elev= 30
       0  696.34    47.6  690.65    99.2  688.29   111.1  685.47   130.9  676.96
   150.8  676.26   186.6  678.02   230.6  677.55   282.5  679.34   310.4  674.59
   334.4  674.13   362.4  671.08   382.4  667.02   422.3  665.14   438.3  661.36
   446.3  660.99   454.3   660.1   466.2  660.88   490.2  660.85   502.2  665.94
   530.2  666.43   554.1  671.22  601.78674.0424  687.83 678.211  758.48682.2859
  776.11682.8489  789.82682.7997  852.51683.4056  883.85682.4824   889.7  682.38
#Mann= 10 ,-1 , 0
       0     .12       0   446.3    .045       0   466.2     .12       0
  601.78     .06       0  687.83     .12       0  758.48     .08       0
  776.11     .06       0  789.82     .08       0  852.51    .016       0
  883.85     .06       0
Bank Sta=446.3,466.2
XS Rating Curve= 0 ,0
Exp/Cntr=0.3,0.1

Type RM Length L Ch R = 1 ,646.3   ,296.7,312.2,325.3
XS GIS Cut Line= 4
     1724507.386      401889.616     1724616.525      402026.214
     1724911.832      402361.645     1725011.658      402539.596
#Sta/Elev= 30
       0  679.36    15.9   678.4    47.7  673.34    63.6  671.84    91.4  670.96
   103.3  669.03   115.2  669.52   139.1  666.72   174.8  666.31   282.6  665.74
   330.5  667.36   382.3  667.69   406.3  665.01   418.2  665.63   422.2  665.24
   434.2  660.36   438.2  658.96   442.2   658.8   454.2  659.06   462.1  661.07
   474.1  664.67     510  665.52     526  666.82   569.9  674.92   585.8  677.26
   609.8  679.36   700.2  683.48   715.9  683.76   766.9  680.92   825.8  680.58
#Mann= 5 ,-1 , 0
       0     .12       0   115.2     .09       0   434.2    .045       0
   462.1     .12       0   569.9     .05       0
#XS Ineff= 2 , 0
       0     350     675               0
Permanent Ineff=
       F       F
Bank Sta=434.2,462.1
XS Rating Curve= 0 ,0
Exp/Cntr=0.3,0.1

Type RM Length L Ch R = 1 ,334.1   ,163.4,135.9,108.9
XS GIS Cut Line= 4
     1724418.989       401793.32     1724451.762      402092.548
     1724518.926      402253.741     1724756.229      402377.955
#Sta/Elev= 30
       0  679.58    15.8  673.34    31.7  668.55    51.5  667.34   130.7  666.97
   227.7 670.267  249.68670.9118   289.1  671.82   332.8  671.62   376.4  670.16
   384.4  668.76   400.2  660.12   404.2  659.12   412.1  657.54     424  657.27
     428  657.31     432  659.05   439.9  664.09   451.8  665.31   487.6  666.98
   511.6  666.27   551.6  667.04   583.6  665.74   603.6  666.27   627.6  668.69
   647.5  672.48   703.5  679.23   715.5  681.73   735.5  688.81   743.5  690.48
#Mann= 7 ,-1 , 0
       0     .12       0    51.5     .05       0   227.7    .045       0
  249.68     .12       0   384.4    .012       0   404.2    .045       0
   647.5     .08       0
#XS Ineff= 2 , 0
       0     305     675     551       0     675
Permanent Ineff=
       F       F
Bank Sta=404.2,432
XS Rating Curve= 0 ,0
Exp/Cntr=0.3,0.1

Type RM Length L Ch R = 1 ,198.2   ,168.8,150.2,131.2
XS GIS Cut Line= 3
       1724267.3      402151.142     1724311.329      402243.198
     1724506.015      402339.944
#Sta/Elev= 30
       0  673.12    31.4  673.19    62.8  674.09    70.6  673.98    82.4   674.8
    98.1  674.26     110   674.7   129.7  673.82   141.6   673.9   145.5   673.2
   149.5  671.09   153.4  668.54   157.4  667.11     185  662.08     189  660.98
  191.85 659.897   196.9  658.12   200.9  657.61   204.8  657.93   208.8  658.67
   212.7  659.86   220.6  662.41   228.5  664.33   240.4  665.21   252.2  667.36
   260.2   667.6   279.9  667.48   291.8  668.37   303.6  667.36   319.4  666.79
#Mann= 3 ,-1 , 0
       0     .12       0  191.85    .045       0   212.7     .12       0
#XS Ineff= 2 , 0
                          292.49          668.88
Permanent Ineff=
       F       F
Bank Sta=191.85,212.7
XS Rating Curve= 0 ,0
Exp/Cntr=0.3,0.1

Type RM Length L Ch R = 1 ,48      ,55,48,40.8
XS GIS Cut Line= 4
     1724332.947      402353.145     1724354.648      402435.611
     1724507.643       402431.27     1724535.855      402374.847
#Sta/Elev= 30
       0  671.62     7.8  671.16    23.3  669.68    27.1  669.11    34.9  666.96
    42.6  664.39    50.4  660.19    54.3  659.13    58.1  658.56   62.75658.3027
    72.7658.1066    81.4  658.06    89.2  658.73    93.1  658.72   136.3   657.6
     152  657.16   155.9  657.29   159.8  658.13   179.5   663.3   187.3  665.88
   191.2  666.77   195.2  667.34   206.9   667.5   218.7  667.12   234.4  667.94
   254.1  667.87     262  667.48   265.9  667.58   289.6  666.09   301.4  666.04
#Mann= 5 ,-1 , 0
       0     .12       0   62.75     .04       0    72.7     .12       0
   136.3    .045       0   159.8     .12       0
#XS Ineff= 2 , 0
       0    89.2  668.04  197.69       0  668.04
Permanent Ineff=
       F       F
Bank Sta=136.3,159.8
XS Rating Curve= 0 ,0
Exp/Cntr=0.3,0.1

Chan Stop Cuts=-1
Use User Specified Reach Order=0
Composite Channel Slope=5
